--- RghthndFrk.prj (project) ---

Proj Title=RghthndFrk
Current Plan=p01
Default Exp/Contr=0,0
English Units
Geom File=g01
Flow File=f01
Plan File=p01
BEGIN DESCRIPTION:
END DESCRIPTION:
DSS Export Rating Curves= 0
DSS Export Rating Curve Sorted= 0
DSS Export Volume Flow Curves= 0
DXF OffsetX= 0
DXF OffsetY= 0
DXF ScaleX= 0
DXF ScaleY= 0

--- RghthndFrk.p01 (plan) ---

Plan Title=Floodplain
Program Version=4.00
Geom File=g01
Flow File=f01
K Sum by GR=0
Std Step Tol=0.01
Critical Tol=0.01
Num of Std Step Trials=20
Max Error Tol=0.3
Flow Tol Ratio=0.001
Split Flow NTrial=30
Split Flow Tol=0.02
Split Flow Ratio=0.02
Log Output Level=0
Friction Slope Method=1
Unsteady Friction Slope Method=2
Unsteady Bridges Friction Slope Method=1
Global Log Level=0
CheckData=False
Run HTab=0
Run UNet=0
Run PostProcess=0
UNET Theta=0
UNET Theta Warmup=0
UNET ZTol=0
UNET ZSATol=0
UNET MxIter=0
UNET MaxInSteps=0
UNET DtIC=0
UNET DtMin=0
UNET MaxCRTS=0
UNET WFStab=0
UNET SFStab=0
UNET WFX=0
UNET SFX=0
UNET DSS MLevel=0
UNET DZMax Abort=0
UNET Convert EG Bridges=0
UNET Use Existing IB Tables=0
UNET Froude Limit=0
UNET Froude Power=0
Write IC File=0
Echo Input=False
Echo Output=False
Write Detailed=0

--- RghthndFrk.f01 (steady flow) ---

Flow Title=NFF Regression Equation
Program Version=4.10
Number of Profiles= 1
Profile Names=P100yr
River Rch & RM=RghthndFrk,Main            ,28923
492.1333
River Rch & RM=RghthndFrk,Main            ,28518
626.0708
River Rch & RM=RghthndFrk,Main            ,28118
661.3199
River Rch & RM=RghthndFrk,Main            ,24889.2
722.8619
River Rch & RM=RghthndFrk,Main            ,21439.6
799.8558
River Rch & RM=RghthndFrk,Main            ,21173.2
1156.502
River Rch & RM=RghthndFrk,Main            ,19712.3
1261.887
River Rch & RM=RghthndFrk,Main            ,14912.3
1382.934
River Rch & RM=RghthndFrk,Main            ,7664.8
1532.993
River Rch & RM=RghthndFrk,Main            ,7192.7
1891.912
River Rch & RM=RghthndFrk,Main            ,1341.6
2013.587
River Rch & RM=RghthndFrk,Main            ,822.5
    2502
Boundary for River Rch & Prof#=RghthndFrk,Main            , 1
Up Type= 0
Dn Type= 1
Dn Known WS=2370.1
DSS Import GetInterval= 0
DSS Import GetPeak= 0
DSS Import FillOption= 0

--- RghthndFrk.g01 (geometry) ---

Geom Title=USGS 3m DEM
Program Version=4.10

River Reach=RghthndFrk      ,Main
Reach XY= 30
     1892775.604       172509.63     1893450.083      172017.442
     1894314.667      170604.682     1894859.425      168727.207
     1897707.896      165880.723     1897756.073      164025.255
     1898112.844      163477.078     1897942.271      163010.932
     1898082.896      161957.546     1897597.219      161289.578
     1897795.136      160702.338     1897240.448      160158.067
     1897495.656      158948.432     1896905.813      158441.921
     1896455.292      157564.317     1895379.852      157311.489
     1895338.104      157758.327     1894706.594      157796.088
     1895072.513      156880.234     1894413.625      156273.953
      1894172.74      155462.755     1894433.157        154991.4
     1894039.927      154501.817     1894921.731      153755.515
     1894868.735      153463.553     1894355.031      153202.338
     1894426.594      152876.767     1894604.091      152708.663
     1895046.471      152832.394     1895312.426      152372.753

Type RM Length L Ch R = 1 ,28923   ,394.4,405,418.4
XS GIS Cut Line= 3
     1893110.014      172746.189     1892743.765      172480.368
     1892307.792      172459.508
#Sta/Elev= 30
       0 2636.38    49.2 2603.79      59 2592.97    68.9 2584.43    88.5    2571
    98.4 2565.74   137.7 2553.32   167.2 2539.15   177.1 2529.54   186.9 2523.09
   255.8 2484.75   275.5 2469.06     305 2453.65   324.6 2447.37     402 2445.98
   403.4 2445.96     417 2446.62   442.7 2451.08   472.4    2449   492.2 2452.28
   531.9 2460.34   551.8 2467.78   611.3 2480.64   631.1 2486.76     641 2488.32
   760.1 2500.68   809.7 2508.22   849.3 2508.35   859.3 2509.67     889 2516.85
#Mann= 3 , 0 , 0
       0     .08       0     402    .045       0     417     .08       0
Bank Sta=402,417
XS Rating Curve= 0 ,0
Exp/Cntr=0.3,0.1

Type RM Length L Ch R = 1 ,28518   ,403.9,400,391.2
XS GIS Cut Line= 3
     1893238.386      172620.028     1893047.559      172221.061
     1892919.892      171838.059
#Sta/Elev= 30
       0 2644.76      59 2612.48    78.6 2608.57   127.8 2584.35   176.9 2554.21
   186.7 2552.72   196.6 2547.62     226 2529.27   275.2 2494.29   294.8 2487.32
   334.2  2463.1   363.6 2447.84   373.5 2443.66   383.3 2442.38   432.4  2442.3
   434.8  2442.3   449.8 2442.41   511.2 2449.68   540.7 2468.63   599.8 2501.72
   609.6 2503.29   639.2 2515.29   658.9 2517.83   668.7 2522.21   698.3 2544.03
   708.1 2546.53   727.8 2563.34   796.7 2614.76   816.4  2622.2     846 2640.96
#Mann= 3 , 0 , 0
       0     .08       0   434.8    .045       0   449.8     .08       0
Bank Sta=434.8,449.8
XS Rating Curve= 0 ,0
Exp/Cntr=0.3,0.1

Type RM Length L Ch R = 1 ,28118   ,406.9,400,394.9
XS GIS Cut Line= 3
     1893647.349      172383.606       1893391.7      172065.253
     1893106.201      171762.241
#Sta/Elev= 30
       0 2507.78      10 2504.86    29.9 2501.88    59.8 2501.43    79.7 2499.22
   129.5 2487.62   149.4 2486.21   159.3 2482.61   189.2 2476.01     239 2470.92
     249 2472.22   258.9 2470.91   298.8 2457.93   318.7 2454.49   338.6 2448.04
   400.8 2440.16   415.8 2438.61   507.4  2438.1     557 2442.86   566.9 2444.87
   576.8 2448.82   646.2 2492.91     666  2498.5   675.9 2502.92   685.8 2510.17
   705.7 2522.18   735.4 2537.33     785 2558.91   804.8 2564.21   824.6 2574.12
#Mann= 3 , 0 , 0
       0     .08       0   400.8    .045       0   415.8     .08       0
Bank Sta=400.8,415.8
XS Rating Curve= 0 ,0
Exp/Cntr=0.3,0.1

Type RM Length L Ch R = 1 ,27718   ,396.8,400,401.8
XS GIS Cut Line= 3
       1893944.1      171960.617     1893603.377      171733.466
     1893262.653      171506.315
#Sta/Elev= 30
       0 2651.26      10 2644.08      20 2634.88    99.9  2586.6   109.9 2577.88
   119.8 2572.66   159.8 2558.17   169.8 2553.21   199.8 2535.48   209.7 2526.46
   219.7 2520.78   309.6 2474.23   329.6 2467.26   379.5 2442.25     402 2435.23
     417 2433.85   419.5 2433.78   499.4 2435.87   529.4 2437.54   549.3 2440.08
   599.3 2457.65   619.2 2467.43   649.2 2478.62   679.2 2480.39   689.2  2482.4
   699.2 2487.02   719.1 2499.88     789 2537.83     799 2543.74     819 2557.93
#Mann= 3 , 0 , 0
       0     .08       0     402    .045       0     417     .08       0
Bank Sta=402,417
XS Rating Curve= 0 ,0
Exp/Cntr=0.3,0.1

Type RM Length L Ch R = 1 ,27318   ,413.2,405.8,400
XS GIS Cut Line= 3
     1894152.594      171688.351     1893846.628      171416.382
     1893525.552      171161.015
#Sta/Elev= 30
       0 2588.48    49.9 2574.75    89.9 2561.64   119.8 2559.35   129.8 2559.58
   139.8 2557.99   149.8  2554.3   189.7  2534.9   209.7 2519.93   259.6 2493.03
   269.6 2488.21   289.6 2482.68   319.5 2466.08   379.4 2438.09   389.4 2433.77
   401.9 2430.98   409.4  2430.3   416.9 2430.37   516.8 2432.41   536.4 2434.24
   585.2    2454   604.7 2459.08   624.3 2460.07   663.3 2485.22   673.1 2488.21
   692.6 2487.96   721.9 2483.92   731.7 2485.43     761 2493.67   819.6 2502.35
#Mann= 3 , 0 , 0
       0     .08       0   401.9    .045       0   416.9     .08       0
Bank Sta=401.9,416.9
XS Rating Curve= 0 ,0
Exp/Cntr=0.3,0.1

Type RM Length L Ch R = 1 ,26912.2 ,393,394,394.8
XS GIS Cut Line= 3
     1894396.678      171221.092     1893842.735      170984.538
     1893577.119      170883.019
#Sta/Elev= 30
       0 2620.14     9.9 2607.91    49.4 2576.13    59.2 2570.47    69.1 2567.72
   138.2 2563.46   167.9 2555.78     237 2508.45   256.7 2498.38   266.6 2490.16
   276.5  2484.8   345.6 2454.21   355.5 2446.32   385.1 2433.82   404.8 2427.79
   420.1 2426.43   424.6 2426.29   435.1 2426.49   464.1 2428.97   513.5 2428.53
     553 2438.64   592.5 2442.85   602.3 2447.39     622 2461.76   700.4 2501.24
   710.2 2508.49   729.8 2518.79   798.4 2549.21   827.9 2557.73   886.7 2580.89
#Mann= 3 , 0 , 0
       0     .08       0   420.1    .045       0   435.1     .08       0
Bank Sta=420.1,435.1
XS Rating Curve= 0 ,0
Exp/Cntr=0.3,0.1

Type RM Length L Ch R = 1 ,26518   ,210.7,204.1,197.3
XS GIS Cut Line= 3
     1894585.617      170950.489     1894226.892      170761.688
     1893846.144      170555.754
#Sta/Elev= 30
       0 2559.22    19.8 2556.94    49.4 2557.92      89 2547.97   118.6 2535.45
   148.3  2517.3     178 2502.93   237.3 2481.93   257.1  2480.2     267 2478.01
   306.5 2466.13   316.4    2461   326.3 2453.73     346 2441.97   365.8 2431.26
   385.6 2424.81   395.5 2423.81   397.9 2423.84   412.9 2424.85     425 2428.34
   434.9 2429.23   493.9  2429.5   513.6  2431.8   582.5 2458.87   602.1 2469.34
   661.2 2494.79   680.8 2500.79   690.7 2505.98   759.5 2534.98   838.2 2576.89
#Mann= 3 , 0 , 0
       0     .08       0   397.9    .045       0   412.9     .08       0
Bank Sta=397.9,412.9
XS Rating Curve= 0 ,0
Exp/Cntr=0.3,0.1

Type RM Length L Ch R = 1 ,26313.9 ,129.5,125.7,121.9
XS GIS Cut Line= 2
     1894556.724      170628.473     1893852.122      170489.407
#Sta/Elev= 30
       0 2536.25      10 2529.19      20 2519.77    69.8 2503.34    89.8 2495.44
    99.8 2486.38   169.6 2453.63   179.6 2444.79   189.5 2439.46   219.4 2426.13
   232.7  2423.9   239.4 2423.75   247.7 2423.77   269.3 2428.52   279.3  2428.9
   319.2 2426.81   339.2 2427.32   349.1 2429.34   359.1 2433.14     409 2458.66
   428.9 2472.88   468.8 2489.67   488.8 2499.63   508.7  2512.8   588.5 2548.42
   598.5 2556.25   668.3 2586.69   678.3  2593.3   688.3 2598.17   718.2 2610.94
#Mann= 3 , 0 , 0
       0     .08       0   232.7    .045       0   247.7     .08       0
#XS Ineff= 2 , 0
                          279.26          2428.9
Permanent Ineff=
       F       F
Bank Sta=232.7,247.7
XS Rating Curve= 0 ,0
Exp/Cntr=0.3,0.1

Type RM Length L Ch R = 1 ,26188.2 ,483.8,500.7,517.4
XS GIS Cut Line= 3
     1894718.852      170458.867     1894464.361      170461.649
     1893869.854      170447.228
#Sta/Elev= 30
       0 2621.17     9.8    2615    19.6 2604.33    97.9 2566.61   127.2 2565.18
   166.4 2543.63   176.2 2535.22     186 2531.48   205.6 2529.24   215.4 2524.74
   254.5 2502.64   274.3 2486.05   333.8 2452.28   353.6 2436.84   383.4  2424.9
     397 2423.83     412 2423.77   432.9 2426.56   492.4 2427.47   502.3 2431.33
   512.2 2440.54   571.7 2475.56   581.6 2482.51   591.5 2493.36   660.9 2531.68
   670.8 2541.43   740.2 2574.23   750.1    2583   799.6 2609.62   849.2 2631.15
#Mann= 3 , 0 , 0
       0     .08       0     397    .045       0     412     .08       0
#XS Ineff= 2 , 0
                          445.45         2433.69
Permanent Ineff=
       F       F
Bank Sta=397,412
XS Rating Curve= 0 ,0
Exp/Cntr=0.3,0.1

Type RM Length L Ch R = 1 ,25687.4 ,346,346.8,347.9
XS GIS Cut Line= 2
     1894764.502      170319.737      1894156.45      169763.343
#Sta/Elev= 30
       0 2562.16    19.9 2558.66    59.6 2562.55    69.5 2560.12    89.4  2552.4
    99.3 2542.93   109.2 2536.19   158.9 2510.75   178.7 2504.36   198.6    2502
     278 2474.63   297.9 2464.17   307.8 2457.77   317.8 2448.36   347.6 2430.44
   357.5 2427.64   401.5 2421.82   416.5 2418.11   417.1 2417.98   486.6 2426.55
   536.2 2440.27     576 2454.66   635.5 2484.16   675.2 2508.98   685.2 2513.22
   695.1 2514.53     705  2519.4   774.6 2554.81   814.3 2579.53   824.2 2582.64
#Mann= 3 , 0 , 0
       0     .08       0   401.5    .045       0   416.5     .08       0
Bank Sta=401.5,416.5
XS Rating Curve= 0 ,0
Exp/Cntr=0.3,0.1

Type RM Length L Ch R = 1 ,25340.6 ,459.9,451.3,438.5
XS GIS Cut Line= 3
     1895010.829      170017.447     1894646.861      169790.843
     1894283.025       169585.49
#Sta/Elev= 30
       0 2491.28    19.9 2484.87    69.8 2471.48    99.7  2466.6   179.5  2449.6
   199.4 2446.07   239.3 2443.58   259.2 2441.23   279.2 2442.56   309.1 2437.33
     339 2429.17   368.9 2426.82   388.9 2419.23   403.5 2417.25   418.5 2416.62
   418.8 2416.61   478.5  2422.2   488.4  2424.6   498.4 2429.07   558.1 2468.33
     568 2476.78     578 2486.58   617.7 2511.18   657.5 2533.18   677.4 2546.13
   697.3 2553.25     757 2583.74     767 2591.23   776.9 2597.51   846.5 2634.74
#Mann= 3 , 0 , 0
       0     .08       0   403.5    .045       0   418.5     .08       0
Bank Sta=403.5,418.5
XS Rating Curve= 0 ,0
Exp/Cntr=0.3,0.1

Type RM Length L Ch R = 1 ,24889.2 ,297.1,294.8,292.5
XS GIS Cut Line= 2
     1895148.298      169460.065     1894332.956       169350.82
#Sta/Elev= 30
       0 2573.23     9.9 2572.61    59.5  2553.2    99.1  2531.1   118.9 2523.34
   148.7 2515.52     228  2483.1   267.6 2460.47   287.4 2443.91   297.3 2439.53
   317.2  2437.4   366.7 2422.56   403.4 2415.41   406.4 2414.92   418.4 2415.31
   436.1 2419.22   465.8 2430.52   485.6 2444.98   545.1 2477.68     555 2484.35
   564.9 2496.51   634.3 2542.15   644.2 2554.48   713.6 2595.14   723.5 2603.81
   733.4 2609.28   753.2 2616.25     783 2617.72   792.9 2615.53   822.6  2600.7
#Mann= 3 , 0 , 0
       0     .08       0   403.4    .045       0   418.4     .08       0
Bank Sta=403.4,418.4
XS Rating Curve= 0 ,0
Exp/Cntr=0.3,0.1

Type RM Length L Ch R = 1 ,24594.4 ,496.9,510.8,524.7
XS GIS Cut Line= 2
     1895183.664      169121.775      1894351.07      169110.024
#Sta/Elev= 30
       0 2566.83    39.6  2547.8    49.6 2545.88     109 2526.57   128.9 2515.27
   158.6  2503.6   188.3 2487.72   208.2 2469.36   237.9  2451.6   247.8 2448.13
   267.6 2446.79   277.6    2443   287.5 2434.35   317.2 2417.44   327.1 2414.53
     337 2413.84   399.6 2416.45   414.6 2417.06   436.2 2418.16   446.1 2420.62
   495.6 2439.58   515.5 2448.67   525.4 2457.17   594.8 2489.29   604.7 2498.39
   654.2 2521.24   674.1 2527.86   743.5 2526.55   783.1 2520.92   832.7    2516
#Mann= 3 , 0 , 0
       0     .08       0   399.6    .045       0   414.6     .08       0
Bank Sta=399.6,414.6
XS Rating Curve= 0 ,0
Exp/Cntr=0.3,0.1

Type RM Length L Ch R = 1 ,24083.1 ,364.8,376,387.1
XS GIS Cut Line= 2
     1895255.878      168912.092     1894579.669      168437.182
#Sta/Elev= 30
       0 2597.25    19.9 2595.73    39.8 2591.31    59.7 2584.06    69.7 2578.64
    79.6 2571.23    99.6 2552.22   109.5 2544.77   129.4 2536.33   179.2  2528.3
   209.1 2520.42     229  2513.2   278.8 2484.82   308.6 2466.23   328.5 2451.34
   338.5 2447.16   358.4 2445.04   368.4  2440.4   398.2 2418.82   408.2 2413.54
   420.8 2412.25   435.8 2412.18   537.6 2411.88   557.5 2414.69   577.4    2423
   627.2 2451.41   647.1 2467.56     677 2484.32   746.7 2514.76   826.3 2530.08
#Mann= 3 , 0 , 0
       0      .1       0   420.8    .045       0   435.8      .1       0
Bank Sta=420.8,435.8
XS Rating Curve= 0 ,0
Exp/Cntr=0.3,0.1

Type RM Length L Ch R = 1 ,23707.1 ,401.3,394.4,385.8
XS GIS Cut Line= 3
     1895369.918      168786.901      1895093.52      168264.374
     1894908.918      168090.208
#Sta/Elev= 30
       0 2572.06    29.6 2558.17    59.1 2547.33    78.8 2545.09   118.2 2534.34
   177.3 2522.46   187.2 2522.89   206.9 2516.97   236.4 2502.79   275.9 2480.16
   295.6 2473.25   305.4 2463.98   315.3 2450.01   325.1  2441.1   344.8 2441.02
   354.7 2438.62   364.5 2432.66   384.2 2415.62   394.1 2411.33   398.8 2411.27
   413.8  2411.3   502.5 2409.77     532 2412.44   551.7 2418.32   639.9 2471.23
   659.5 2479.15   688.7 2498.53   757.1 2537.95   786.4 2560.38   844.9 2583.71
#Mann= 3 , 0 , 0
       0      .1       0   398.8    .045       0   413.8      .1       0
Bank Sta=398.8,413.8
XS Rating Curve= 0 ,0
Exp/Cntr=0.3,0.1

Type RM Length L Ch R = 1 ,23312.3 ,399.8,399.9,398.5
XS GIS Cut Line= 3
     1895720.171      168413.716      1895413.73      168135.608
     1895092.905      167880.828
#Sta/Elev= 30
       0 2553.44     9.8  2549.4    88.7 2534.14   118.2 2523.65   206.9 2472.75
   226.6 2459.34   246.3 2440.46   256.2 2435.22   285.7 2432.56   295.6  2429.5
   325.2 2412.21     335 2409.62   406.3 2407.99   421.3  2407.8   423.8 2407.79
   453.8 2412.22   513.8 2441.34   553.7 2463.04   573.7 2476.52   583.7 2479.09
   593.7 2484.93   653.6 2521.86   683.6 2543.49   713.6 2560.24   733.6 2566.67
   753.6 2576.62   763.6 2579.12   793.5 2593.18   803.5 2596.11   823.5 2595.72
#Mann= 3 , 0 , 0
       0      .1       0   406.3    .045       0   421.3      .1       0
Bank Sta=406.3,421.3
XS Rating Curve= 0 ,0
Exp/Cntr=0.3,0.1

Type RM Length L Ch R = 1 ,22912.3 ,403.4,399.9,400.1
XS GIS Cut Line= 3
     1895994.915        168165.6     1895697.253      167875.911
     1895369.754      167622.548
#Sta/Elev= 30
       0 2493.11    59.3  2477.5    79.1  2471.3   108.8 2464.96   148.3 2453.47
   168.1 2447.05   187.9 2437.64   227.5 2428.06   237.4 2426.29   257.1 2425.29
     267 2423.29   296.7 2411.18   336.2 2408.09   407.9 2406.57   415.4 2406.47
   422.9 2406.71   523.8 2414.33   533.7 2416.59   543.5  2419.9   573.1 2431.14
   602.7 2441.43   622.4 2442.66   632.2 2444.24     652 2445.47     721 2454.53
   740.7 2456.38   770.3 2462.22   780.1 2460.69     790 2460.78   829.4 2467.89
#Mann= 3 , 0 , 0
       0      .1       0   407.9    .045       0   422.9      .1       0
Bank Sta=407.9,422.9
XS Rating Curve= 0 ,0
Exp/Cntr=0.3,0.1

Type RM Length L Ch R = 1 ,22512.3 ,417.3,421.5,424.8
XS GIS Cut Line= 3
      1896299.86      167884.559     1895974.096      167629.246
     1895662.762      167364.416
#Sta/Elev= 30
       0 2567.99    39.4 2561.25    88.7 2543.83   118.2 2531.09     138 2520.28
   157.7 2505.04   167.5 2499.71   187.2 2492.87   246.4 2458.29   256.2 2452.11
   266.1  2443.1   305.5 2420.02   315.4 2417.47   344.9 2416.65   374.5 2406.28
   394.2 2405.84   406.4 2405.92   421.4 2406.51   463.7 2412.34   503.6 2431.08
   563.4 2467.85   583.4 2486.25   623.2 2513.09   643.2 2525.58   663.1 2534.08
   683.1 2546.18   762.8 2576.05   772.8 2576.93   792.7 2583.22   822.6 2597.13
#Mann= 3 , 0 , 0
       0      .1       0   406.4    .045       0   421.4      .1       0
Bank Sta=406.4,421.4
XS Rating Curve= 0 ,0
Exp/Cntr=0.3,0.1

Type RM Length L Ch R = 1 ,22090.7 ,648.4,651,653.7
XS GIS Cut Line= 4
     1896965.969      169281.179     1896825.379      168611.635
     1896487.035      167580.039     1895993.492      167021.929
#Sta/Elev= 30
       0 2467.14    59.5 2462.52   138.8 2440.02   267.7 2470.21   446.2 2492.92
   525.5 2480.53   644.5 2501.15   753.9 2501.97   803.7 2495.48   953.1 2496.94
  1042.7 2471.89  1092.5 2464.82  1192.1 2484.95  1331.6 2490.82  1441.1 2503.75
  1490.9 2518.84  1560.6 2509.23  1590.5 2510.53  1809.5 2538.76  1839.4 2527.03
  1869.2 2505.68    1889 2484.88  1968.5 2430.92  2008.2 2414.43    2094 2402.67
  2097.6 2402.33    2109  2403.1  2206.9 2428.64  2405.6 2520.02  2514.8 2539.31
#Mann= 3 , 0 , 0
       0      .1       0    2094    .045       0    2109      .1       0
Bank Sta=2094,2109
XS Rating Curve= 0 ,0
Exp/Cntr=0.3,0.1

Type RM Length L Ch R = 1 ,21439.6 ,274.1,266.4,258
XS GIS Cut Line= 4
     1897206.605      169165.806     1897201.386      168361.143
     1896889.415      167119.505     1896555.786      166654.521
#Sta/Elev= 30
       0 2470.92    69.5 2476.06   168.9  2471.5     298 2486.07   596.1 2496.62
     755 2516.36   844.4  2506.4   923.8 2471.77   983.3 2426.73  1052.8 2419.85
  1112.3 2431.33  1181.8  2462.1  1231.4 2475.78  1380.3 2515.41  1410.1 2517.49
  1509.3 2502.26  1608.6 2462.46  1787.2 2499.29  1886.4 2502.75  2025.4 2493.47
  2173.7 2424.49    2223 2409.99  2279.4 2404.69  2294.4 2401.57  2311.8  2400.9
  2371.1 2406.32  2430.3 2426.09  2489.5 2450.77  2588.1 2509.58  2657.2 2532.33
#Mann= 3 , 0 , 0
       0      .1       0  2279.4    .045       0  2294.4      .1       0
Bank Sta=2279.4,2294.4
XS Rating Curve= 0 ,0
Exp/Cntr=0.3,0.1

Type RM Length L Ch R = 1 ,21173.2 ,258.2,260.8,264
XS GIS Cut Line= 3
     1897268.736      166996.305     1896931.194      166753.678
     1896582.316      166524.774
#Sta/Elev= 30
       0 2545.51    59.4 2522.25   108.9 2497.87   118.8 2494.17   128.7 2492.74
   138.6  2488.1   168.3 2468.93   207.8 2446.84   227.6  2437.1   247.4 2429.25
   267.2 2426.27   306.8 2415.81   346.4 2413.98   405.8 2402.34   418.5 2401.05
   425.6  2400.8   433.5 2401.08   445.5 2402.54   465.4 2407.23   475.3  2414.8
   485.2 2419.36   495.2 2422.41   554.8 2456.36   574.6 2470.73   584.6 2473.39
   654.1 2510.93     674 2518.09   773.4 2571.23   783.3 2574.77     833 2586.71
#Mann= 3 , 0 , 0
       0      .1       0   418.5    .045       0   433.5      .1       0
Bank Sta=418.5,433.5
XS Rating Curve= 0 ,0
Exp/Cntr=0.3,0.1

Type RM Length L Ch R = 1 ,20912.3 ,171,170.3,169.5
XS GIS Cut Line= 3
     1897408.433      166826.124     1897098.377      166558.624
     1896788.322      166291.125
#Sta/Elev= 30
       0 2569.47      20 2567.38      40 2562.16    49.9 2555.06   139.8 2513.34
   189.8 2488.22   259.7 2439.39   279.7  2421.9   289.6 2419.74   319.6 2418.55
   369.6 2408.32   389.5 2401.55     402  2400.5   409.5 2400.42     417 2400.74
   469.4 2405.92   499.4 2416.83   529.4 2431.61   549.3 2444.33   579.3  2466.8
   599.3 2489.28   609.3 2496.88   629.2 2508.83   659.2 2531.94   689.2 2552.32
   699.2 2561.36   729.1 2569.89   759.1    2571     799 2575.19     819 2573.63
#Mann= 3 , 0 , 0
       0      .1       0     402    .045       0     417      .1       0
Bank Sta=402,417
XS Rating Curve= 0 ,0
Exp/Cntr=0.3,0.1

Type RM Length L Ch R = 1 ,20742.2 ,581.2,581.4,581.6
XS GIS Cut Line= 4
     1897880.098      166911.491     1897581.202      166702.399
     1897328.777      166525.815     1896962.879      166231.612
#Sta/Elev= 30
       0 2502.46    49.3 2499.73   108.4 2486.83     138 2489.46   147.9 2487.62
   246.5 2449.83     276 2443.54   295.8 2442.52   364.8 2463.98   434.3 2492.67
   523.8 2503.92   543.6 2509.45   553.6 2508.99   573.5 2503.35   613.2 2485.66
   623.1 2479.28     643 2459.21   662.9 2448.69   702.8 2421.76   722.8 2420.26
   823.2 2400.59   832.7 2400.55   838.2 2400.89   902.6 2409.62   942.6 2431.24
  1012.5 2457.87  1042.4 2466.47  1062.4  2476.6  1112.4 2489.36  1142.3 2491.95
#Mann= 3 , 0 , 0
       0      .1       0   823.2    .045       0   838.2      .1       0
Bank Sta=823.2,838.2
XS Rating Curve= 0 ,0
Exp/Cntr=0.3,0.1

Type RM Length L Ch R = 1 ,20160.6 ,463.7,448.2,433.2
XS GIS Cut Line= 3
     1898050.685      166637.068     1897689.731      166085.747
     1897275.323       165751.93
#Sta/Elev= 30
       0 2446.37    99.8 2468.37   119.8    2469   169.7 2479.38   219.7 2487.09
   239.6 2484.45   329.5 2499.23   349.4  2497.5   369.4 2498.79   389.4 2495.38
   439.3 2493.15   479.2 2485.26   509.2 2475.89   539.2 2461.39   599.1 2441.95
   678.7 2410.59   718.1 2407.36   774.4 2398.99   777.2  2398.7   789.4 2400.81
   875.8  2435.9   895.5 2450.68   974.3 2494.44     994 2511.88  1013.7 2523.21
  1043.3  2535.8  1092.6 2560.41  1112.3 2572.21  1171.4 2598.12  1191.1  2604.8
#Mann= 3 , 0 , 0
       0      .1       0   774.4    .045       0   789.4      .1       0
Bank Sta=774.4,789.4
XS Rating Curve= 0 ,0
Exp/Cntr=0.3,0.1

Type RM Length L Ch R = 1 ,19712.3 ,317.7,319.1,320
XS GIS Cut Line= 3
     1898119.236       165607.21     1897709.368      165605.805
     1897300.057      165597.281
#Sta/Elev= 30
       0 2574.12      30 2567.99      50  2561.5      60 2551.72     130 2515.61
     140 2505.15   209.9  2469.1   219.9 2459.42   249.9 2440.62   259.9 2436.04
   289.9 2426.46   299.9 2419.58   319.9 2412.64   369.9 2407.53   379.9 2402.82
   402.4  2398.3   409.9 2398.28   417.4 2399.26   449.8 2406.94   459.8 2415.29
   529.7 2448.13   539.7 2457.86   609.6 2497.43   619.6 2509.32   689.5 2551.11
   699.4 2560.23   709.4 2564.48   719.4 2566.23   769.3 2564.67   819.3 2577.88
#Mann= 3 , 0 , 0
       0      .1       0   402.4    .045       0   417.4      .1       0
Bank Sta=402.4,417.4
XS Rating Curve= 0 ,0
Exp/Cntr=0.3,0.1

Type RM Length L Ch R = 1 ,19393.3 ,477,483.9,490.9
XS GIS Cut Line= 3
     1898344.888      165438.008      1897850.43       165299.56
     1897293.342      165265.571
#Sta/Elev= 30
       0 2495.28   118.5 2495.42   148.1 2496.84   177.7 2501.66   296.2 2505.61
   385.1    2496   404.8 2490.18   454.2 2471.75   464.1 2464.24   483.8 2454.12
   543.4 2431.87   553.3 2424.02   573.3 2414.86   593.2 2409.61   623.1 2407.24
   633.1 2400.92   646.5 2397.22     653 2396.73   661.5 2397.08   702.8 2402.02
   722.8 2406.67   742.7 2414.65   782.6 2435.33   792.5 2442.62   802.5 2445.86
   882.2 2450.51   971.9 2453.02  1021.8 2458.18  1041.7 2462.93  1071.6  2467.2
#Mann= 3 , 0 , 0
       0      .1       0   646.5    .045       0   661.5      .1       0
Bank Sta=646.5,661.5
XS Rating Curve= 0 ,0
Exp/Cntr=0.3,0.1

Type RM Length L Ch R = 1 ,18909.2 ,411.7,396.9,382.2
XS GIS Cut Line= 3
     1898443.779      165279.781     1897978.989      164906.466
     1897464.111      164699.406
#Sta/Elev= 30
       0 2443.33    69.6 2451.78   109.3 2452.39     149 2448.71   288.1 2456.01
     308 2451.48   397.4 2455.57   437.2 2450.42   486.9  2451.5   526.6 2442.71
   576.3 2436.04   606.1 2428.46   625.9 2419.72   665.5 2410.83   695.2 2408.56
   713.4 2402.46   728.4 2397.61   734.9 2397.13   754.7  2401.6   794.4 2419.04
   863.7 2442.77   883.5 2457.74   952.9 2499.69   962.8 2509.07  1022.3 2538.19
    1052 2547.42  1071.8 2548.27  1121.4 2547.08  1131.3    2545  1151.1 2535.43
#Mann= 3 , 0 , 0
       0      .1       0   713.4    .045       0   728.4      .1       0
Bank Sta=713.4,728.4
XS Rating Curve= 0 ,0
Exp/Cntr=0.3,0.1

Type RM Length L Ch R = 1 ,18512.3 ,481.8,495.9,510.1
XS GIS Cut Line= 3
     1898254.964      164359.426      1897860.57      164469.625
     1897466.176      164579.824
#Sta/Elev= 30
       0 2440.46      20 2442.13   119.8 2459.32   179.8 2473.27   199.8  2475.2
   219.7 2469.16   239.7 2456.79   299.6 2433.44   309.6 2428.58   319.6 2421.66
   339.6  2413.7   359.6 2408.42   379.5 2407.83   389.5 2404.46   399.5 2396.37
     402  2396.1   409.5 2395.31     417 2396.33   459.4  2405.9   469.4 2409.45
   489.4 2420.36   549.3 2443.06   569.3  2452.3   609.3 2463.94   619.2 2465.18
   679.2 2465.62   719.1 2464.87   739.1  2462.7     779 2462.31     819 2463.66
#Mann= 3 , 0 , 0
       0      .1       0     402    .045       0     417      .1       0
Bank Sta=402,417
XS Rating Curve= 0 ,0
Exp/Cntr=0.3,0.1

Type RM Length L Ch R = 1 ,18016.3 ,295.4,303.9,310.1
XS GIS Cut Line= 3
     1898207.381       164148.87     1897553.756      163922.495
     1897427.669       163873.05
#Sta/Elev= 30
       0 2513.02    19.8 2508.11    29.6  2503.6    98.8 2495.66   118.6 2490.23
   187.8 2481.82   197.6  2475.6     247 2457.69   266.8 2448.87   286.6 2435.55
   345.9 2410.01   355.7 2407.73   385.4 2405.16   451.7  2393.9   454.6 2393.61
   466.7 2395.52   484.2 2399.84   523.7 2403.71   543.5 2412.51   573.1 2422.59
   592.9 2431.64   612.7 2441.72   622.5 2451.92     672 2480.78   691.7 2494.46
   711.1  2514.3   740.1 2532.84   798.1 2565.06   817.5 2571.42   827.2 2573.41
#Mann= 3 , 0 , 0
       0      .1       0   451.7    .045       0   466.7      .1       0
Bank Sta=451.7,466.7
XS Rating Curve= 0 ,0
Exp/Cntr=0.3,0.1

Type RM Length L Ch R = 1 ,17712.3 ,437.3,419.9,404.8
XS GIS Cut Line= 3
     1898278.877      164030.983     1897967.667      163765.878
      1897628.03       163530.25
#Sta/Elev= 30
       0  2575.1      10 2571.64    29.9 2561.77   119.6 2530.96   159.5 2513.48
   219.4 2481.53   239.3 2466.53   259.2 2455.02   279.2 2447.81     339 2412.97
     349 2408.29   368.9 2406.29   388.9 2397.75   401.3 2394.08   408.8 2393.59
   416.3 2394.89     458 2403.56   467.9  2408.5   536.8 2456.06   556.4  2473.7
     586 2491.84   595.8 2496.89   635.2 2510.68   654.9 2520.07   684.4 2529.39
   694.2 2530.24   704.1 2528.28     773 2496.96   802.5 2495.04   822.2 2487.52
#Mann= 3 , 0 , 0
       0      .1       0   401.3    .045       0   416.3      .1       0
Bank Sta=401.3,416.3
XS Rating Curve= 0 ,0
Exp/Cntr=0.3,0.1

Type RM Length L Ch R = 1 ,17292.4 ,432.5,432.7,429.6
XS GIS Cut Line= 2
     1898505.115      163358.463     1897664.121        163423.8
#Sta/Elev= 30
       0 2494.12    19.8 2497.64    39.7 2504.38    59.5 2503.47   168.7  2507.1
   178.6 2505.87   248.1 2469.21     258 2462.98   267.9 2452.49   337.4 2416.18
   347.3 2407.46   377.1 2405.16   398.9  2395.5   413.9 2393.35   416.8 2393.32
   436.6 2399.81   476.4 2400.59   496.2 2405.81   506.1 2414.89   575.6 2451.94
   585.5 2461.17   595.4  2467.6   615.3 2476.79   625.2 2478.85   694.7 2483.78
   734.4 2472.46   754.2  2461.3   793.9 2448.22   823.7  2443.7   843.5 2444.55
#Mann= 3 , 0 , 0
       0      .1       0   398.9    .045       0   413.9      .1       0
Bank Sta=398.9,413.9
XS Rating Curve= 0 ,0
Exp/Cntr=0.3,0.1

Type RM Length L Ch R = 1 ,16859.2 ,335.4,346.7,359.9
XS GIS Cut Line= 3
     1898362.255      162907.324      1897936.62       163034.67
     1897543.866      163133.836
#Sta/Elev= 30
       0 2530.03    39.5  2515.5    59.2  2505.2   128.4 2479.04   138.2  2472.2
   148.1 2468.08   177.7 2456.52   207.3 2447.03   227.1 2437.27   286.3 2417.44
   315.9 2404.49   325.8 2401.62   365.3  2399.2     385 2396.09   429.4 2391.84
   434.4 2391.72   444.4 2392.16   454.2 2394.35     464 2399.43   533.2 2425.72
   543.1 2433.44   612.2 2464.04     632 2476.79   641.9 2479.73   671.5  2483.8
   691.3 2484.09     711 2481.83   780.2 2486.35   819.7 2486.16   849.4 2488.44
#Mann= 3 , 0 , 0
       0     .06       0   429.4    .045       0   444.4     .06       0
Bank Sta=429.4,444.4
XS Rating Curve= 0 ,0
Exp/Cntr=0.3,0.1

Type RM Length L Ch R = 1 ,16512.3 ,402.6,400,397.1
XS GIS Cut Line= 3
     1898386.966      162838.159      1897961.54      162693.494
     1897576.488      162576.689
#Sta/Elev= 30
       0 2543.74    69.9 2519.28    79.9 2512.62    89.9 2508.13   149.8 2486.17
   169.8 2474.98   239.6 2449.72   249.6 2442.44   259.6 2438.04   319.5 2415.98
   339.5 2406.35   379.4  2402.7   409.4 2397.29   419.4 2393.67   439.4 2391.49
   441.8 2391.62   456.8 2393.81   488.6  2403.6   508.2 2414.38   567.1  2440.3
   576.9 2445.32   586.8 2455.21   616.2 2471.38   655.4 2491.19   675.1 2504.19
   743.8 2531.96   753.6 2538.28   763.4 2542.28   832.1 2564.14   851.7 2571.99
#Mann= 3 , 0 , 0
       0     .06       0   441.8    .045       0   456.8     .06       0
Bank Sta=441.8,456.8
XS Rating Curve= 0 ,0
Exp/Cntr=0.3,0.1

Type RM Length L Ch R = 1 ,16112.3 ,489.6,477.8,463.1
XS GIS Cut Line= 3
     1898547.971      162343.465     1898142.401      162354.139
     1897713.706      162309.868
#Sta/Elev= 30
       0 2571.53    29.7 2564.09    69.3  2548.4    79.2 2540.44   108.8 2528.51
   118.7 2528.54   158.3 2512.89   168.2  2505.1   237.5 2474.15   247.4 2465.11
   316.6 2426.18   326.6 2415.79   336.4 2408.74   346.3 2404.48     376 2401.02
   398.2 2394.19   413.2 2392.03   415.5 2391.99   454.7  2401.1   474.3 2413.37
   493.9 2432.09   552.6 2464.85   572.2 2480.18   591.8 2489.79   640.8 2507.94
   650.6 2514.35   728.9 2540.55   758.3 2548.59   777.9 2549.79   836.7 2545.85
#Mann= 3 , 0 , 0
       0     .06       0   398.2    .045       0   413.2     .06       0
Bank Sta=398.2,413.2
XS Rating Curve= 0 ,0
Exp/Cntr=0.3,0.1

Type RM Length L Ch R = 1 ,15634.3 ,321.9,317.9,313.9
XS GIS Cut Line= 3
     1898443.779      161670.241      1898315.22      161732.048
     1897674.709      162131.515
#Sta/Elev= 30
       0 2591.84      19 2589.33    47.6 2583.01    66.6 2579.77    85.6 2573.88
   123.6 2563.98   162.5 2549.76   172.4 2543.11   212.2 2523.32   251.9 2500.38
   351.2 2434.22   361.2 2424.36     381 2412.51     391 2407.61   400.9 2404.86
   420.8 2402.94   450.6 2392.23   460.5 2391.83   465.6 2392.22   500.2  2396.4
   539.9 2399.15   609.5  2425.6   629.3  2426.6   669.1 2431.12   708.8 2432.28
   738.6 2437.78   798.2 2451.14     818 2448.67   837.9 2449.44   897.5 2459.05
#Mann= 3 , 0 , 0
       0     .06       0   450.6    .045       0   465.6     .06       0
Bank Sta=450.6,465.6
XS Rating Curve= 0 ,0
Exp/Cntr=0.3,0.1

Type RM Length L Ch R = 1 ,15316.3 ,389.4,403.7,414.3
XS GIS Cut Line= 3
     1898117.879      161412.479     1897635.341      161848.246
     1897452.392      161961.971
#Sta/Elev= 30
       0 2551.01    88.7 2542.97    98.5 2538.86   108.4 2531.71   128.1  2524.6
   137.9 2519.31     197 2483.58   216.7 2468.75   246.3 2450.67     266 2444.18
   325.1 2406.72   354.6 2403.94   407.8 2392.73   422.8  2391.6   423.6 2391.55
   443.3 2393.18   472.9 2398.98   512.3 2423.67     532 2437.93   551.7 2446.01
   610.8 2476.92   650.2 2505.87   669.8 2517.21   689.4 2525.39   708.9 2530.31
   748.1 2532.62   767.7 2530.08   797.1 2530.95   826.4 2535.93   865.6 2545.92
#Mann= 3 , 0 , 0
       0     .06       0   407.8    .045       0   422.8     .06       0
Bank Sta=407.8,422.8
XS Rating Curve= 0 ,0
Exp/Cntr=0.3,0.1

Type RM Length L Ch R = 1 ,14912.3 ,366.3,379.3,396.1
XS GIS Cut Line= 3
     1898068.475      161314.093     1897617.765      161361.714
     1897230.931      161470.299
#Sta/Elev= 30
       0 2541.45    59.1  2533.4   128.1 2531.69   147.8 2529.04   157.6 2526.47
   177.4 2518.32     197 2499.95   236.5 2468.24   256.2 2453.65   275.9 2435.61
   315.3 2415.87     335 2408.04     404 2397.95   433.5 2391.66   443.4 2391.49
   445.7 2391.49   460.7 2391.77   502.2 2395.78   521.8 2405.72     561 2421.25
   580.6 2431.11   590.4 2438.41   600.2 2447.92   639.4 2472.36   668.8 2488.77
   678.6 2497.74   688.4  2503.5   747.2 2532.58   766.8  2545.6     855  2581.6
#Mann= 3 , 0 , 0
       0      .1       0   445.7    .045       0   460.7      .1       0
Bank Sta=445.7,460.7
XS Rating Curve= 0 ,0
Exp/Cntr=0.3,0.1

Type RM Length L Ch R = 1 ,14533.1 ,473.2,452.2,431.2
XS GIS Cut Line= 3
     1898094.637      161202.739     1897566.117      160935.972
      1897312.27         160909.
#Sta/Elev= 30
       0 2527.32     9.9 2526.43    49.3 2517.93    78.9 2508.65   128.3 2495.67
     148 2488.74   167.7 2478.57   207.2 2463.03   236.8 2453.05   256.6 2440.78
   325.6 2412.48   335.5 2409.16   365.1 2404.24     398 2392.86     413 2391.67
   424.3 2394.24   434.2 2399.28   463.8  2408.1   513.1 2426.04     523 2432.25
   552.6 2444.26     592 2462.07   601.8 2468.02   611.7 2476.14   680.4 2507.21
   690.2 2514.48   758.9 2539.96   768.8 2546.08   778.6 2549.58   847.3 2569.98
#Mann= 3 , 0 , 0
       0     .08       0     398    .045       0     413     .08       0
Bank Sta=398,413
XS Rating Curve= 0 ,0
Exp/Cntr=0.3,0.1

Type RM Length L Ch R = 1 ,14080.8 ,326.9,320.5,314.6
XS GIS Cut Line= 2
     1898095.187      160431.625     1897308.673      160802.713
#Sta/Elev= 30
       0  2472.4      10 2471.52      30 2474.15      50 2473.98     130 2460.46
     140 2457.45   159.9 2447.81   169.9 2435.01   179.9 2424.77   189.9 2417.34
   199.9 2413.07   299.9 2404.86   359.9 2401.69   396.6  2391.8   399.8 2391.38
   411.6 2391.85   449.8 2399.77   469.8 2408.66   509.8 2432.15   529.8 2448.75
   579.8 2478.18   599.8 2491.94   619.8 2512.12   639.8 2522.85   669.7    2533
   709.7  2544.1   779.7 2560.36   789.7 2565.41   799.7 2568.39   869.7 2578.36
#Mann= 3 , 0 , 0
       0     .08       0   396.6    .045       0   411.6     .08       0
Bank Sta=396.6,411.6
XS Rating Curve= 0 ,0
Exp/Cntr=0.3,0.1

Type RM Length L Ch R = 1 ,13760.2 ,511.7,531,549.7
XS GIS Cut Line= 2
       1897842.4       160122.46     1897193.422      160680.003
#Sta/Elev= 30
       0 2512.41      10 2513.47    29.8 2505.96   129.3 2450.34   149.2 2446.08
   179.1 2427.87     199 2413.82   208.9 2411.42   228.8 2402.84   248.7 2400.27
   348.2 2400.43   430.8 2391.09   445.8 2390.52   447.7  2390.5   497.4 2393.97
   507.4 2395.35   517.3 2399.52   567.1 2440.08     587 2454.73   606.9 2463.98
   636.7  2481.3   676.5 2502.43   696.4 2510.46   706.4 2512.39   726.2 2512.59
   736.2 2512.15   746.2 2509.93   805.8 2512.18   825.7 2509.97   855.6 2511.38
#Mann= 3 , 0 , 0
       0     .08       0   430.8    .045       0   445.8     .08       0
Bank Sta=430.8,445.8
XS Rating Curve= 0 ,0
Exp/Cntr=0.3,0.1

Type RM Length L Ch R = 1 ,13229.2 ,310.3,316.9,325.9
XS GIS Cut Line= 3
     1897794.365      160007.324     1897479.587      160045.948
     1896882.178      159953.108
#Sta/Elev= 30
       0  2527.7    79.3 2515.45    99.1 2510.16   118.9 2501.61   188.3 2481.06
   198.2 2474.79   237.8 2456.99   257.7 2445.54   267.6 2438.54   277.5 2425.06
   307.2 2405.75   317.1 2401.04     327 2399.19   515.4 2390.65   521.4 2390.84
   536.4 2391.93     555 2394.68   564.9 2398.22   584.7 2407.68   604.6 2421.42
     664 2448.96   683.8 2461.43   693.8 2465.54   753.2 2486.64   763.1 2491.99
   832.5 2513.26   862.2 2525.27   901.9 2536.78   911.8 2540.68   921.7 2548.36
#Mann= 3 , 0 , 0
       0     .08       0   521.4    .045       0   536.4     .08       0
Bank Sta=521.4,536.4
XS Rating Curve= 0 ,0
Exp/Cntr=0.3,0.1

Type RM Length L Ch R = 1 ,12912.3 ,379.9,371.8,361.4
XS GIS Cut Line= 3
      1897831.14      159940.835     1897461.477      159768.817
     1897096.505      159551.324
#Sta/Elev= 30
       0 2543.31    29.8 2533.83    69.6 2523.83    79.6 2519.78   149.2 2498.58
   159.1 2493.95   169.1 2486.74   198.9 2473.47   228.7 2457.43   248.6 2443.95
   258.6 2434.53   288.4 2418.29   348.1 2397.94   377.9 2396.41   400.2 2392.23
   415.2  2390.7   417.6 2390.59   457.1  2394.8   506.5 2412.02   516.4 2416.09
   526.3 2425.51   536.2 2431.73   565.8 2446.94   605.3 2464.26   625.1 2476.33
     714 2508.28   723.9 2514.74     803  2541.1   822.7 2550.98   832.6 2554.11
#Mann= 3 , 0 , 0
       0     .08       0   400.2    .045       0   415.2     .08       0
Bank Sta=400.2,415.2
XS Rating Curve= 0 ,0
Exp/Cntr=0.3,0.1

Type RM Length L Ch R = 1 ,12540.5 ,455.3,441.8,428.2
XS GIS Cut Line= 2
     1897938.101      159439.261     1897088.965      159373.486
#Sta/Elev= 30
       0 2539.51    19.8 2532.91    29.7 2527.03      99 2504.37   108.9 2497.57
   178.3 2475.19   188.2 2469.98   217.9 2458.81   257.5 2441.71   267.4 2433.63
   277.3 2427.72   326.8 2405.72   336.7 2402.98   366.4 2399.61   402.3 2390.72
     406 2390.25   417.3 2391.84   435.7 2394.25   465.4 2393.14   495.2 2402.16
     515 2412.52   574.4 2435.39   594.2 2449.16   653.6 2479.73   663.5 2485.99
   673.4 2494.26   742.7 2520.68   752.6 2527.34   812.1  2548.4   851.7 2550.11
#Mann= 3 , 0 , 0
       0     .08       0   402.3    .045       0   417.3     .08       0
Bank Sta=402.3,417.3
XS Rating Curve= 0 ,0
Exp/Cntr=0.3,0.1

Type RM Length L Ch R = 1 ,12098.7 ,392.8,386.2,385.5
XS GIS Cut Line= 3
     1897904.299       158954.41     1897682.314      158896.334
     1897078.631      159231.772
#Sta/Elev= 30
       0  2578.4    29.9 2574.16    59.9  2566.4    79.8 2558.22    89.8 2550.33
   159.6 2524.48   169.6 2516.39   229.5 2489.32   239.3 2482.51     259 2462.75
     338 2411.11   347.8 2403.29   387.3 2399.82   397.2 2397.65   418.7 2388.14
   426.8 2386.14   433.7 2386.58   466.2 2389.65     486 2394.19   535.3 2421.01
   604.4 2446.02   624.1 2457.48   683.3 2485.14     703  2492.7   722.8  2495.2
   752.4 2494.56   811.6 2499.31     851 2503.16   900.3 2510.93   920.1 2511.33
#Mann= 3 , 0 , 0
       0     .08       0   418.7    .045       0   433.7     .08       0
Bank Sta=418.7,433.7
XS Rating Curve= 0 ,0
Exp/Cntr=0.3,0.1

Type RM Length L Ch R = 1 ,11712.3 ,403.4,399.7,385.1
XS GIS Cut Line= 3
     1897520.107      158484.571     1897209.495      158792.791
     1896861.187      158998.553
#Sta/Elev= 30
       0 2524.09    19.9 2522.92    29.8 2519.63    49.7 2506.61    89.5 2483.61
   109.4 2475.92   139.2 2456.99   159.1 2440.45     179 2433.01   218.8 2408.22
   228.7 2403.74   268.5 2397.52   288.4 2396.99   338.1 2390.82   430.1 2384.52
   445.1 2383.85   447.4  2383.8   457.3 2384.96   467.2 2388.34   486.9 2400.59
   526.4 2418.93   546.1 2425.93     556 2431.22   565.8 2439.99   654.7 2494.42
   713.9 2515.54   733.6 2520.07   753.3 2530.42   802.7 2550.53   842.1 2561.16
#Mann= 3 , 0 , 0
       0     .08       0   430.1    .045       0   445.1     .08       0
Bank Sta=430.1,445.1
XS Rating Curve= 0 ,0
Exp/Cntr=0.3,0.1

Type RM Length L Ch R = 1 ,11312.3 ,397.5,399.9,405.4
XS GIS Cut Line= 3
     1897275.366       158160.17     1896993.187      158504.938
     1896754.665       158835.75
#Sta/Elev= 30
       0 2492.75     9.9 2493.62    19.8 2492.27    49.5 2484.36   108.9  2459.6
   118.8 2457.01   128.7 2456.99   138.6 2452.97   168.3 2439.68     198 2423.46
   247.5 2409.35   257.4 2408.35   306.9 2394.13   326.7  2393.5   425.7  2383.1
     438 2383.74     453 2386.66   475.4 2392.11   485.3 2396.49   505.2  2402.1
     535 2416.97   554.9 2430.74   574.8  2437.4   604.7 2450.94   674.3 2474.38
   694.2 2483.93   773.8 2500.44   793.7 2498.62   823.5  2503.4   853.4 2512.01
#Mann= 3 , 0 , 0
       0     .08       0     438    .045       0     453     .08       0
Bank Sta=438,453
XS Rating Curve= 0 ,0
Exp/Cntr=0.3,0.1

Type RM Length L Ch R = 1 ,10912.3 ,386,396.8,407.3
XS GIS Cut Line= 3
     1897122.213      157972.201     1896787.769       158223.17
     1896458.394      158464.531
#Sta/Elev= 30
       0 2564.09    39.8 2554.27    69.7 2539.76   129.4 2501.98   139.4 2498.05
   159.3 2482.75   238.9 2436.43   258.8 2420.33   298.7 2398.83   318.6 2392.93
   348.4 2390.71   398.2 2381.73   408.2 2381.39   410.6 2381.47   425.6 2382.94
     448 2388.56   527.7 2391.69   537.6 2393.86   547.6 2398.04   567.5 2413.39
   597.4 2431.34   607.4 2435.88   617.3  2439.5   637.2 2443.42   667.1 2453.87
     687 2458.65   716.9 2462.29   746.8  2463.8   786.6 2460.61   826.5 2463.33
#Mann= 3 , 0 , 0
       0     .08       0   410.6    .045       0   425.6     .08       0
Bank Sta=410.6,425.6
XS Rating Curve= 0 ,0
Exp/Cntr=0.3,0.1

Type RM Length L Ch R = 1 ,10515.5 ,433.3,404.4,375.6
XS GIS Cut Line= 3
     1897062.918      157782.803     1896517.867      157875.279
     1896253.332      157939.559
#Sta/Elev= 30
       0  2529.4    59.2 2504.15      79 2492.58   138.2 2466.78     158 2455.88
   187.6 2447.28   217.2 2432.85   236.9  2426.9   246.8 2422.52   266.6 2411.57
   276.4 2410.74     306 2395.45   315.9 2391.63   325.8 2390.22   365.3 2388.98
   400.5 2382.38   404.8  2381.7   415.5  2382.4   473.9 2401.23   493.6 2410.66
   562.6 2433.82   572.3 2442.13   591.7 2455.42   611.2 2472.44   620.9 2479.59
   659.8 2501.46     689 2511.96   747.3 2527.96   776.5 2525.28   825.1 2523.61
#Mann= 3 , 0 , 0
       0      .1       0   400.5    .045       0   415.5      .1       0
Bank Sta=400.5,415.5
XS Rating Curve= 0 ,0
Exp/Cntr=0.3,0.1

Type RM Length L Ch R = 1 ,10111   ,398.4,398.7,398.9
XS GIS Cut Line= 3
      1896485.56         157162.     1896399.197      157768.971
     1896204.077      157947.952
#Sta/Elev= 30
       0 2559.75     9.9 2559.48    39.6 2548.71    69.2 2533.56    98.9 2512.32
   108.8 2512.66   187.9 2448.21   197.8  2447.3   217.6 2439.05   247.2 2431.94
   286.8  2406.3   316.4 2395.77   346.1  2392.3   385.6 2381.44   395.2 2380.91
   395.5 2380.89   410.2 2381.37   454.9 2387.82   484.5 2399.84   494.4 2400.91
   583.4 2449.08   593.3 2449.17   613.1 2459.56   681.7 2476.35   701.3 2478.47
     721 2478.23   740.6 2481.51   779.8 2495.15   848.4 2523.99   877.9 2527.53
#Mann= 3 , 0 , 0
       0      .1       0   395.2    .045       0   410.2      .1       0
Bank Sta=395.2,410.2
XS Rating Curve= 0 ,0
Exp/Cntr=0.3,0.1

Type RM Length L Ch R = 1 ,9712.3  ,384.3,387.1,389.9
XS GIS Cut Line= 3
     1896096.202      157102.166     1896033.934      157506.905
     1895971.667      157911.643
#Sta/Elev= 30
       0 2533.79      40  2515.4    59.9 2509.16    89.9 2491.19   139.8 2456.08
   149.8 2450.86   219.7 2443.86   229.7  2440.8   239.7 2435.55   249.7 2434.86
   269.7 2422.81   299.6 2401.07   309.6 2396.88   349.6  2392.7   369.6 2388.21
   389.5 2381.15   399.5 2379.69     402 2379.75     417 2381.22   429.5 2383.34
   489.4 2385.62   499.4 2387.29   529.4 2402.47   549.3 2408.42   629.2 2449.42
   649.2  2454.5   709.1 2484.98   729.1  2492.9     779 2499.89     819  2500.5
#Mann= 3 , 0 , 0
       0      .1       0     402    .045       0     417      .1       0
Bank Sta=402,417
XS Rating Curve= 0 ,0
Exp/Cntr=0.3,0.1

Type RM Length L Ch R = 1 ,9325.1  ,757.8,731.9,706.5
XS GIS Cut Line= 3
     1895774.277      157008.736     1895642.677      157494.547
     1895803.834      157883.704
#Sta/Elev= 30
       0 2470.09    49.4 2464.21    59.2 2460.83   118.4 2415.32   138.2 2403.28
   167.8 2399.59   325.7 2399.61   345.4 2396.64   382.3 2379.62   384.9 2378.76
   394.8  2379.5   397.3 2381.58   434.2 2417.23   444.1 2418.99   463.8 2427.44
   483.6 2425.89   493.4 2421.03   522.9 2397.03   532.7 2392.71   552.3 2395.83
   571.9 2407.85   581.7 2410.71     660 2419.13   748.2 2439.15     758 2439.19
   836.4 2469.54     856 2473.84   865.8 2472.25   895.1 2482.86   924.5 2491.09
#Mann= 3 , 0 , 0
       0      .1       0   382.3    .045       0   397.3      .1       0
Bank Sta=382.3,397.3
XS Rating Curve= 0 ,0
Exp/Cntr=0.3,0.1

Type RM Length L Ch R = 1 ,8593.1  ,441.7,460.1,478.4
XS GIS Cut Line= 3
     1895325.334       157133.68     1895180.359      157504.436
     1895622.899      157904.947
#Sta/Elev= 30
       0 2417.28    19.9 2412.49    29.9 2412.67    39.8 2416.53    59.7 2430.72
    79.6 2433.75   119.4  2432.1   179.1 2425.94     199 2426.03   278.7 2437.14
   318.5 2450.06   348.3 2463.66   388.1 2465.05   398.1  2464.1   427.9 2454.16
   527.4 2409.78   547.3 2398.22   557.3 2395.12   666.7 2376.72   686.6 2375.34
   689.2 2375.77   704.2 2379.54   716.4 2383.93   736.3 2388.02   746.3 2392.81
   776.1 2413.08   845.7 2450.53   905.4 2484.82   975.1 2520.85     995 2532.91
#Mann= 3 , 0 , 0
       0      .1       0   689.2    .045       0   704.2      .1       0
Bank Sta=689.2,704.2
XS Rating Curve= 0 ,0
Exp/Cntr=0.3,0.1

Type RM Length L Ch R = 1 ,8132.9  ,432.7,468,503.3
XS GIS Cut Line= 5
     1895325.334       157133.68     1894970.215      157618.161
     1894979.866       157996.49     1894187.942       158811.04
      1894006.64      159453.835
#Sta/Elev= 30
       0 2417.28    29.5 2412.52    98.5 2447.53   167.4 2450.67   236.3 2466.16
   482.5 2468.49   531.8 2460.41   680.4 2400.15   801.6 2373.85   809.8 2373.62
   816.6 2374.73   919.4 2402.74   989.1 2442.32    1029 2453.62  1198.4 2408.06
    1318 2455.78  1357.8 2459.33  1457.5 2447.86  1527.2 2452.63  1567.1 2443.03
  1716.6  2432.6  1786.4 2412.82  1836.2 2429.95  1905.9 2473.13  1925.9 2478.78
  2145.1 2452.39  2374.4 2462.89  2523.9 2442.35  2643.5 2397.53  2783.1 2395.63
#Mann= 3 , 0 , 0
       0      .1       0   801.6    .045       0   816.6      .1       0
Bank Sta=801.6,816.6
XS Rating Curve= 0 ,0
Exp/Cntr=0.3,0.1

Type RM Length L Ch R = 1 ,7664.8  ,459.2,471.9,483.8
XS GIS Cut Line= 5
     1895460.698      156910.143     1894928.186      157615.689
     1894503.154      157643.495     1893891.734      158700.128
     1893629.754      159289.565
#Sta/Elev= 30
       0 2497.96    19.9 2489.81    79.5 2499.59   109.2 2494.02   198.6  2465.4
   278.1  2413.3   307.9 2417.88   367.5 2456.28   417.1 2464.69   794.6    2467
     874 2429.63  1002.8 2386.01  1104.5 2371.63  1111.8 2371.18  1119.5 2371.99
  1171.2 2390.87  1280.2 2455.77  1359.5  2514.9    1429 2547.16  1518.3 2564.66
  1895.5 2507.01  1945.1 2492.36  2044.3 2439.01  2143.6 2412.52  2242.8 2399.71
    2352 2406.73  2471.1 2445.24    2620 2472.17  3036.8  2480.7  3175.7  2474.2
#Mann= 3 , 0 , 0
       0      .1       0  1104.5    .045       0  1119.5      .1       0
Bank Sta=1104.5,1119.5
XS Rating Curve= 0 ,0
Exp/Cntr=0.3,0.1

Type RM Length L Ch R = 1 ,7192.7  ,713.5,676.7,639.8
XS GIS Cut Line= 3
      1895464.48      156846.485     1895078.995      157331.376
     1894555.113      157025.701
#Sta/Elev= 30
       0 2545.23      50  2529.6    99.9 2519.48   119.9 2520.85   159.9 2512.14
   229.8 2477.47   259.8 2467.84   329.7  2415.8   349.7 2414.65   369.7 2419.53
   419.6 2444.54   459.6 2453.86   569.5 2457.38   609.5 2454.69   639.3 2448.92
   679.1 2435.37   768.6 2397.58   806.1 2375.24   818.3 2371.24   821.1 2371.26
   838.2 2372.67   858.1  2379.3     878 2391.28   957.5 2427.39   997.3 2436.26
    1047 2469.94  1086.8 2513.83  1106.7 2526.23  1156.4 2548.43    1226 2558.79
#Mann= 3 , 0 , 0
       0      .1       0   806.1    .045       0   821.1      .1       0
Bank Sta=806.1,821.1
XS Rating Curve= 0 ,0
Exp/Cntr=0.3,0.1

Type RM Length L Ch R = 1 ,6516.1  ,382.4,385.8,385.9
XS GIS Cut Line= 3
     1895098.731      156307.197     1894782.321      156896.253
     1894514.986      156922.602
#Sta/Elev= 30
       0 2558.07    29.9 2560.46    59.9 2561.26    69.9 2560.05    79.8  2555.1
   149.7 2509.05   159.7 2507.14   169.7 2501.46   189.6 2488.23   209.6 2471.89
   249.5 2445.02   269.5 2437.78   349.3 2384.88   359.3  2379.6   389.2 2375.79
   399.2 2372.04   409.2 2370.28   414.2 2370.78   469.1 2388.04     479 2388.77
   538.9 2409.12   588.8 2412.02   598.8 2420.02   608.8 2434.44   618.8 2444.04
   668.7 2462.46   688.6 2475.68   768.2 2510.13   847.7 2530.79   937.3 2530.48
#Mann= 3 , 0 , 0
       0      .1       0   399.2    .045       0   414.2      .1       0
Bank Sta=399.2,414.2
XS Rating Curve= 0 ,0
Exp/Cntr=0.3,0.1

Type RM Length L Ch R = 1 ,6130.2  ,385.8,399.9,417.4
XS GIS Cut Line= 3
     1894826.614      156136.447     1894577.275      156471.821
     1894382.181      156831.894
#Sta/Elev= 30
       0 2487.72    19.9 2491.11    89.6 2523.35    99.5 2524.99   109.4 2522.45
   159.2 2503.21     209 2477.94   228.8 2466.12   238.8 2455.97   258.7 2446.08
   358.2 2385.66   368.2 2381.31     408 2370.32   410.4 2370.33   417.9 2370.36
   425.4 2373.18   467.8 2397.66   487.8 2403.81   497.8 2408.42   507.8 2410.45
   527.8 2411.85   587.7 2424.64   597.7 2424.93   667.6 2440.27   687.6  2446.1
   697.6 2445.96   707.6 2448.57   797.5 2480.43   817.4 2482.81   827.4 2486.54
#Mann= 3 , 0 , 0
       0      .1       0   410.4    .045       0   425.4      .1       0
Bank Sta=410.4,425.4
XS Rating Curve= 0 ,0
Exp/Cntr=0.3,0.1
